HEC-RAS study LTBLUESTRV.prj: LTBLUESTRV

--- LTBLUESTRV.g01 (geometry) --- (continued)

Type RM Length L Ch R = 1 ,35492   ,60.9,57.2,55.1
XS GIS Cut Line= 4
1963453.34045766228813.7078803321963323.20288022228504.138188536
1963234.47271378228332.5932000891962950.53618118227890.914149374
#Sta/Elev= 30
       0 2049.89   122.7 2041.53   158.3 2033.78   204.6 2029.41   218.8  2030.8
   240.5 2025.55   254.4 2025.33   279.3 2015.92   300.7 2012.17   351.1 1997.18
  376.821983.495   394.1 1980.59  412.261983.492   421.2 1988.39     521 1990.31
   559.5 1995.98     579 2006.12   594.6 2024.32     618 2037.94   644.4 2036.99
   664.8 2043.56   703.7 2046.67   794.6 2046.18   840.3 2051.38   855.9 2056.09
   897.7 2062.19   941.1 2080.61   988.6 2095.88  1031.3 2107.34    1054 2110.48
#Mann= 10 ,-1 , 0
       0      .1       0     220     .04       0  376.82    .045       0
  412.26     .04       0  435.81      .1       0  445.81     .04       0
  548.95      .1       0  628.95     .04       0  788.95     .12       0
  908.95     .04       0
#XS Ineff= 2 , 0
             364 1989.48     424         1989.48
Permanent Ineff=
       F       F
Bank Sta=376.82,412.26
XS Rating Curve= 0 ,0
Exp/Cntr(USF)=0,0
Exp/Cntr=0.5,0.3

Type RM Length L Ch R = 1 ,35435   ,125.9,148.2,163.2
XS GIS Cut Line= 5
1963561.78843887228817.6514432851963469.54918324228635.230301054
1963391.27213493 228496.595046811963312.99508661228371.163150114
1963101.27329116227786.907958501
#Sta/Elev= 30
       0 2027.48    50.3 2023.42      76 2025.48   242.4 2012.34   409.4 1990.49
   413.2 1989.67  422.951983.184   428.7 1980.58   455.8 1980.62  463.831983.184
   482.8 1987.46   490.6 1987.03   502.2 1989.22     524 1988.41     538 1991.05
   558.9 2001.05   572.9  2020.7   632.2  2042.1   691.5 2057.82   764.8 2068.39
   813.7 2066.79   824.1 2068.41   836.1 2065.85   928.8 2077.91   942.8 2085.64
   977.7 2096.72  1016.9 2116.51  1064.9 2133.81  1096.3 2150.88  1132.9 2174.25
#Mann= 13 ,-1 , 0
       0      .1       0      20     .04       0     190      .1       0
  234.42     .04       0  344.42     .12       0  393.62     .04       0
  422.95    .045       0  463.83     .04       0  571.48      .1       0
  681.48     .04       0  891.48      .1       0  901.48     .04       0
 1101.48      .1       0
#XS Ineff= 2 , 0
             4201989.482     465         1989.48
Permanent Ineff=
       F       F
Bank Sta=422.95,463.83
XS Rating Curve= 0 ,0
Exp/Cntr(USF)=0,0
Exp/Cntr=0.5,0.3

Type RM Length L Ch R = 1 ,35286   ,253.8,264.9,292.7
XS GIS Cut Line= 4
1963575.62476094228804.2880468831963486.18475317228521.593736611
1963502.15618313228294.799431194 1963320.0818816227727.813667653
#Sta/Elev= 30
       0 2021.96    29.6  2021.2    67.5  2016.3   139.8 2011.97   184.5 2006.44
   215.3 1998.26   229.2 1991.69   249.9  1986.3   347.3 1983.39  354.631981.212
   403.2 1979.54  408.631981.214   419.7 1987.41   439.4 1989.81   462.3 1999.22
   482.2 2010.26   549.1 2054.54     587 2071.74   604.8 2083.26   642.1  2102.6
   690.4 2122.25   729.1 2130.51   781.3  2136.7   869.5 2160.81   914.4 2170.19
   945.4 2170.79  1007.4  2158.9  1045.3 2155.25  1103.9 2174.58  1119.4 2185.54
#Mann= 5 ,-1 , 0
       0     .04       0  354.63    .045       0  408.63      .1       0
  506.51     .12       0  613.86      .1       0
#XS Ineff= 2 , 0
          333.52 1998.79
Permanent Ineff=
       F       F
Bank Sta=354.63,408.63
XS Rating Curve= 0 ,0
Exp/Cntr(USF)=0,0
Exp/Cntr=0.3,0.1

Type RM Length L Ch R = 1 ,35022   ,276.1,276.9,247.4
XS GIS Cut Line= 4
1963597.98476288228805.8851898791963602.77619187228713.250896118
1963736.93620353 228537.565166571963789.64192239228056.825124807
#Sta/Elev= 30
       0 2017.32      20 2012.79    49.6 2009.83    62.7 2006.27    79.2 2000.48
   101.7 1985.17   118.1 1977.65  158.991975.223   176.6 1973.25  212.311975.222
   221.1 1977.41     296 1978.63   364.4 1984.33   384.2 1990.83   423.8 2008.44
     437  2015.6   446.9 2024.57   460.1 2031.94   470.4 2044.95   512.9 2074.44
   522.8 2083.04     569 2116.41   595.4 2125.49   625.1 2146.46   671.3 2182.11
   674.9  2186.4   681.2 2197.65   698.6 2211.53   747.2 2238.07   797.4 2257.88
#Mann= 7 ,-1 , 0
       0     .04       0  102.76     .12       0  158.99    .045       0
  212.31     .12       0  343.81     .04       0  443.81     .12       0
  743.81      .1       0
#XS Ineff= 2 , 0
          132.72 1981.29  219.27         1980.84
Permanent Ineff=
       F       F
Bank Sta=158.99,212.31
XS Rating Curve= 0 ,0
Exp/Cntr(USF)=0,0
Exp/Cntr=0.3,0.1

Type RM Length L Ch R = 1 ,34745   ,206.4,202.6,191.5
XS GIS Cut Line= 4
 1963786.4476364228997.5423493861963808.80763834  228914.4909136
1963879.08193016228634.9908893191963912.62193308228104.739414683
#Sta/Elev= 30
       0 2036.98    39.1 2014.47   100.2 1986.72   123.9 1972.33   140.8 1968.96
   154.4 1969.18   164.5 1967.78   208.6 1969.43   249.1 1971.72     266 1970.05
   316.7 1975.36   347.2 1981.87   362.7 1982.16   374.2 1986.92   390.7  1989.7
   407.5 1995.21     426 2004.37   449.9 2007.01   459.7 2013.01   479.4 2018.86
   499.2 2029.18   518.8 2043.13   535.3 2057.44   581.3 2087.21     627 2112.61
   699.7 2148.47   755.6 2185.26     772 2199.53   890.4 2262.47   905.5 2268.39
#Mann= 7 ,-1 , 0
       0      .1       0   154.4    .045       0   208.6      .1       0
  306.01     .12       0  346.01     .04       0  504.21     .12       0
  894.21      .1       0
#XS Ineff= 2 , 0
                          247.61         1973.23
Permanent Ineff=
       F       F
Bank Sta=154.4,208.6
XS Rating Curve= 0 ,0
Exp/Cntr(USF)=0,0
Exp/Cntr=0.3,0.1

Type RM Length L Ch R = 1 ,34542   ,275.5,298.7,318.5
XS GIS Cut Line= 4
1964011.64479882229083.7880711641964027.61622878228924.073771575
1964032.40765777228553.5365965291964054.76765971228222.927996379
#Sta/Elev= 30
       0 2052.63    12.5 2049.26    52.1 2032.63    85.1 2021.52   131.2 1997.52
   200.3 1965.64   223.2 1958.53   236.4 1956.29  253.441958.529   262.8 1964.16
   288.9 1971.03   315.1 1980.72   328.2 1987.06   341.4 1986.88   354.5 1993.27
   390.6 2000.43   452.9 2016.15   479.2 2021.15   498.4 2027.59     525 2032.66
   548.1 2042.38   607.3 2058.83     634 2068.11   692.8 2103.26   715.8 2120.85
   725.7 2122.46   748.7 2139.52   784.9 2160.97   834.2 2192.61   862.4 2207.24
#Mann= 6 ,-1 , 0
       0      .1       0   223.2    .045       0  253.44      .1       0
  280.51     .04       0  480.51     .12       0  771.08      .1       0
Bank Sta=223.2,253.44
XS Rating Curve= 0 ,0
Exp/Cntr(USF)=0,0
Exp/Cntr=0.3,0.1

Type RM Length L Ch R = 1 ,34243   ,311.9,320.2,325.5
XS GIS Cut Line= 4
1964067.54480368229093.3709291391964209.69053031228975.182347444
 1964367.8076869228844.2166217811964364.61340091 228646.17089029
#Sta/Elev= 30
       0 2028.11     9.8 2022.69    49.9 2006.08    78.1 1996.28    97.9 1990.93
   146.3 1979.38   193.3 1972.28     240 1962.55   260.5 1961.21     282 1957.72
   291.3  1955.6  304.981950.494   321.1 1947.71   329.6 1948.59  334.711950.492
   342.4 1954.29   347.2 1958.28   361.2 1992.16   363.3 1996.79   365.9 2000.53
     385 2015.18   412.1 2015.43   422.3 2019.45   455.4 2026.38   491.2 2031.92
   504.3 2037.32   543.7 2038.56   556.8  2040.1   569.9 2037.44   588.2 2036.81
#Mann= 6 ,-1 , 0
       0      .1       0     130     .12       0  294.86     .04       0
  304.98    .045       0  334.71     .04       0  530.17     .12       0
Bank Sta=304.98,334.71
XS Rating Curve= 0 ,0
Exp/Cntr(USF)=0,0
Exp/Cntr=0.3,0.1

Type RM Length L Ch R = 1 ,33923   ,225.7,195.8,170.5
XS GIS Cut Line= 4
1964081.91909064229193.9909378811964158.58195444229184.408079905
1964340.65625597229136.4937900281964433.29054974228927.268057567
#Sta/Elev= 30
       0 2037.64      36 2011.74    52.6 1998.88    85.9 1976.05    96.1 1968.17
   102.9 1961.04   116.4 1943.79   119.8 1940.67  122.451939.632     130  1938.3
   153.8  1937.4  163.39 1939.63   167.3 1942.38   170.7 1943.62   182.1 1945.58
   203.6 1946.22     217 1950.41   219.7 1952.32   231.8 1965.86   235.2 1967.69
   258.9  1976.4   286.6 1983.95   304.5 1986.98   338.9 1990.61   351.2 1993.06
     405 2007.21     432 2006.71   441.9 2007.98   473.2 2014.35   494.3 2014.47
#Mann= 6 ,-1 , 0
       0      .1       0  122.45    .045       0  163.39      .1       0
  187.26     .12       0  325.53      .1       0  415.53     .04       0
Bank Sta=122.45,163.39
XS Rating Curve= 0 ,0
Exp/Cntr(USF)=0,0
Exp/Cntr=0.3,0.1

Type RM Length L Ch R = 1 ,33727   ,207.7,185.6,168
XS GIS Cut Line= 4
1964263.99339217229494.2538211081964283.15910812229404.813813338
1964351.83625695229217.9480828191964444.47055071228944.836630522
#Sta/Elev= 30
       0 2081.23    25.8 2063.78      40 2052.68      50 2040.73    56.8 2034.98
    63.5 2027.32    73.5 2012.54    80.2 1998.13   107.4  1976.5   125.5 1960.14
   142.7 1946.36   149.7 1938.71  154.951934.796   160.2 1933.08   174.1 1932.88
   188.1 1933.18  192.481934.795   205.6 1941.75   223.1 1948.91   275.5 1950.65
   289.5 1952.26   313.8 1957.73   358.4 1973.53   395.7 1981.85   424.6  1990.3
   493.2 2004.97   514.7 2002.88   521.6 2003.47   552.5 2010.11     579 2010.93
#Mann= 6 ,-1 , 0
       0      .1       0  154.95    .045       0  192.48      .1       0
  310.56     .12       0  420.56      .1       0  520.56     .04       0
Bank Sta=154.95,192.48
XS Rating Curve= 0 ,0
Exp/Cntr(USF)=0,0
Exp/Cntr=0.3,0.1

Type RM Length L Ch R = 1 ,33542   ,288,268.6,252.4
XS GIS Cut Line= 4
1964553.07627443229492.656678112 1964524.3277005229392.036669371
1964454.05340868 229201.97665286 1964447.6648367228967.196632464
#Sta/Elev= 30
       0 2118.77    25.3 2098.37   100.4 2043.16   114.3 2028.45   128.3 2011.93
   131.8 2006.78   135.3 1999.16   138.8 1993.88   205.2 1936.92   212.2 1932.17
  219.461929.275   226.2 1927.25   239.2 1926.88  251.571929.274   267.3 1936.65
   271.7 1937.55   340.3 1937.58   352.7 1941.05   372.5 1950.26   382.2  1955.7
     392 1965.51   398.6 1970.15   421.6 1980.45   431.4 1982.99   477.4  1999.5
   483.9 1999.95   493.8 1998.52   503.3 1999.35   523.3 2006.16   542.1    2008
#Mann= 6 ,-1 , 0
       0      .1       0  219.46    .045       0  251.57      .1       0
  307.28     .12       0  407.28      .1       0  507.28     .04       0
Bank Sta=219.46,251.57
XS Rating Curve= 0 ,0
Exp/Cntr(USF)=0,0
Exp/Cntr=0.3,0.1

Type RM Length L Ch R = 1 ,33273   ,305.5,301.4,291.4
XS GIS Cut Line= 4
1964850.14487166 229229.128083791964754.31629191229126.910932053
1964553.07627443 229003.930921371964490.78769759228965.599489468
#Sta/Elev= 30
       0 2092.02      23 2077.07    44.3 2061.29    58.7 2053.43   108.4 2015.89
   116.3 2010.87   126.1 2002.88   135.5 1997.19   159.1 1978.85   171.1 1970.61
   190.2 1954.23   221.6 1934.46   232.5 1924.71   235.5 1923.24  247.191921.215
     253 1919.55   274.8  1919.2   290.4 1920.96   309.4 1921.91   317.1  1925.7
   347.9 1926.31   370.9 1941.34     376 1947.69   390.6 1969.37     394 1972.98
   417.1 1987.12     421 1988.21   428.7 1987.89   436.4  1989.1   449.1 1995.98
#Mann= 4 ,-1 , 0
       0      .1       0  247.19    .045       0   290.4      .1       0
  375.95     .04       0
Bank Sta=247.19,290.4
XS Rating Curve= 0 ,0
Exp/Cntr(USF)=0,0
Exp/Cntr=0.3,0.1

Type RM Length L Ch R = 1 ,32972   ,254,243.6,228.7
XS GIS Cut Line= 4
1964939.25186745228873.6005475161964766.17327119228807.874498302
1964599.66727985228744.3393173961964487.93299618228715.858029403
#Sta/Elev= 30
       0  2023.8    22.5 2015.27    43.6 2003.93    63.9 1990.15    75.1 1981.46
    82.1 1974.94    96.1 1960.42   103.2 1951.47   117.3 1938.13   127.7  1929.6
   138.3 1922.38   150.4 1919.82   194.4 1920.95     219  1920.2   231.8 1917.17
   242.71912.521   254.1 1909.89   275.2 1911.56  277.611912.522   290.2 1920.46
   295.3 1922.75   310.3 1926.72   327.9 1928.47   349.5 1933.38   386.7 1944.94
   400.2 1951.18   413.8 1952.74   436.8 1967.21   456.7 1977.55   478.7  1987.4
#Mann= 4 ,-1 , 0
       0     .12       0   242.7    .045       0  277.61     .12       0
  305.14     .04       0
Bank Sta=242.7,277.61
XS Rating Curve= 0 ,0
Exp/Cntr(USF)=0,0
Exp/Cntr=0.3,0.1

Type RM Length L Ch R = 1 ,32728   ,127.2,99.4,82.8
XS GIS Cut Line= 4
1964887.39401462228610.2800856831964823.50829478228581.886432423
 1964713.4828884228604.9562756971964465.03842237 228571.23881245
#Sta/Elev= 30
       0 1981.57     5.7 1982.25    12.9 1981.33    23.7 1975.43      38 1959.75
    48.8 1951.82    66.7 1932.13    69.8 1930.56    87.1 1908.51    90.4 1905.63
    97.1 1903.86   109.5 1904.43   120.6 1903.12     134 1904.49   144.1 1906.75
   150.8 1911.06   174.2 1916.67   184.3 1916.96   214.1 1914.85   233.9 1919.67
   270.3 1925.55   291.5 1930.64   306.8 1935.81     320 1941.71   333.3 1942.83
     341 1947.84     363 1957.51   376.3 1961.91   412.7 1979.45   433.1 1987.91
#Mann= 6 ,-1 , 0
       0      .1       0      40     .12       0   109.5    .045       0
     134     .12       0  242.33      .1       0  342.33     .12       0
Bank Sta=109.5,134
XS Rating Curve= 0 ,0
Exp/Cntr(USF)=0,0
Exp/Cntr=0.5,0.3

Type RM Length L Ch R = 1 ,32629   ,80.1,83.5,79.1
XS GIS Cut Line= 4
1964887.06529088228478.676841511 1964781.8343104 228433.73624831
  1964717.346179 228531.599875081964463.78094135 228542.22352331
#Sta/Elev= 30
       0 1926.77    12.5 1927.27    32.1 1926.46      66 1920.24    89.6 1912.31
   108.8 1907.79   152.7 1906.58     159 1905.36   163.6 1901.98   170.7 1898.87
   182.5 1898.96   188.5 1897.25   194.1 1897.05   200.4 1898.45   217.9  1904.7
   224.2    1909   240.7 1911.78   260.4 1916.58   326.1 1924.89   342.5 1928.52
   355.9 1932.59   362.2 1934.81   368.8 1938.44   381.9 1939.58     390 1943.75
   411.4 1952.52   424.4 1959.11   437.7 1963.98   456.2 1973.81   485.4 1986.35
#Mann= 6 ,-1 , 0
       0      .1       0      40     .12       0   182.5    .045       0
   200.4     .12       0  291.63      .1       0  391.63     .12       0
#XS Ineff= 2 , 0
           180.5 1898.63  202.67         1898.82
Permanent Ineff=
       F       F
Bank Sta=182.5,200.4
XS Rating Curve= 0 ,0
Exp/Cntr(USF)=0,0
Exp/Cntr=0.5,0.3

Type RM Length L Ch R = 1 ,32545   ,94.8,146.4,188.3
XS GIS Cut Line= 4
1964880.41335041228467.2653129951964767.67232163228388.595968509
1964679.50637713228508.4015464871964475.01535934228516.993912773
#Sta/Elev= 30
       0 1921.56    21.9 1919.13    62.4 1910.06    97.9  1910.3   109.2  1909.1
   131.2 1902.61   137.5  1898.5     146  1897.9   151.81894.414   154.6  1892.5
   171.2 1891.26  182.361894.411   194.9 1900.16   198.9 1901.07   204.5 1900.66
   221.1 1907.67   232.1 1910.45   269.3 1916.24   293.5 1917.06   323.1 1919.77
   369.1 1929.98   386.4 1937.47   398.6 1938.29   401.9  1939.4   408.4 1943.14
   444.6 1957.79   457.7 1965.41   470.9 1970.09   480.4 1975.77   490.9  1980.5
#Mann= 6 ,-1 , 0
       0      .1       0      40     .12       0   151.8    .045       0
  182.36     .12       0  316.23      .1       0  406.23     .12       0
#XS Ineff= 2 , 0
          149.79  1894.4  184.21         1894.45
Permanent Ineff=
       F       F
Bank Sta=151.8,182.36
XS Rating Curve= 0 ,0
Exp/Cntr(USF)=0,0
Exp/Cntr=0.5,0.3

Type RM Length L Ch R = 1 ,32399   ,85.2,97.1,123.4
XS GIS Cut Line= 4
1964881.19256802228462.7873490521964840.59590685228345.911289337
1964735.55235119 228192.47310684 1964624.8204502 228100.99345389
#Sta/Elev= 30
       0 1918.83    12.2 1913.88    22.7 1911.31    33.1 1910.56    50.4 1910.53
    71.3 1906.29    85.2 1907.26   116.4 1906.67   145.5 1901.21   163.1    1892
   166.3 1891.11   173.8 1890.62     179 1889.35   186.9 1888.94   206.6 1890.53
   211.6 1891.65   223.4 1892.52   235.2 1892.01   246.6 1894.09     265 1896.14
     273 1898.57   289.5 1907.59   302.2 1909.01   310.7 1912.16     328 1923.96
   343.3 1932.76     376 1948.45   387.6 1955.91     434 1979.55   453.3 1992.68
#Mann= 6 ,-1 , 0
       0      .1       0      60     .04       0      80     .12       0
   173.8    .045       0   206.6     .12       0  283.73      .1       0
#XS Ineff= 2 , 0
                          227.79         1898.42
Permanent Ineff=
       F       F
Bank Sta=173.8,206.6
XS Rating Curve= 0 ,0
Exp/Cntr(USF)=0,0
Exp/Cntr=0.3,0.1

Type RM Length L Ch R = 1 ,32302   ,64.9,109.2,185.1
XS GIS Cut Line= 4
1964884.52583479228461.5664758371964885.17901677228351.845360183
1964886.34333401228159.733014922 1964946.8878307228030.493800837
#Sta/Elev= 30
       0  1917.5    10.3 1912.62    16.9 1910.83    62.8 1908.95    92.4 1904.93
   108.8 1900.74   161.3 1899.94   174.3 1897.19   194.1 1889.53  201.931888.013
   210.5 1885.68   226.4 1885.22   236.7 1885.47  248.841888.011   253.1 1889.98
   256.4 1892.97   259.7 1900.91   279.4 1902.15   285.9 1907.46   292.5 1910.13
   299.1 1914.44   313.3 1918.72   323.7 1929.02     341 1943.21   374.8  1966.4
   385.7 1975.65   390.4 1977.79   407.5 1979.02   421.9 1994.26   444.6 2010.46
#Mann= 7 ,-1 , 0
       0      .1       0      50     .04       0  149.72     .12       0
  201.93    .045       0  248.84     .12       0  249.72     .04       0
  351.84      .1       0
Bank Sta=201.93,248.84
XS Rating Curve= 0 ,0
Exp/Cntr(USF)=0,0
Exp/Cntr=0.5,0.3

Type RM Length L Ch R = 1 ,32192   ,51.3,50.2,51.5
XS GIS Cut Line= 4
  1964888.325955228460.9795194581964918.94421684228316.915842863
1965035.58621694228354.2791325181965218.50033954 228103.47110992
#Sta/Elev= 30
       0 1916.33    13.3 1910.64    69.4 1908.39    80.4 1906.82   102.6 1897.59
  160.861886.599   177.6 1884.44   201.7    1885  207.211886.599   222.4 1894.11
   232.7 1896.78   249.9 1897.14   263.7  1899.5   327.7 1897.99   339.5 1900.11
   343.5 1901.86   353.6 1908.97     377 1929.33   391.1 1931.76   397.5 1934.84
   409.6 1946.69   422.9 1954.45   450.3  1972.8   475.7 1991.61   490.9 2004.27
   516.1 2021.35   532.8 2034.69   551.8 2047.42   560.2 2054.44   580.2 2064.65
#Mann= 6 ,-1 , 0
       0      .1       0      50     .04       0  160.86    .045       0
  207.21     .04       0  319.76      .1       0  469.76     .12       0
#XS Ineff= 2 , 0
          156.29 1886.62  211.41         1886.72
Permanent Ineff=
       F       F
Bank Sta=160.86,207.21
XS Rating Curve= 0 ,0
Exp/Cntr(USF)=0,0
Exp/Cntr=0.5,0.3

Type RM Length L Ch R = 1 ,32142   ,138.3,113,69.5
XS GIS Cut Line= 4
1964896.27877014228461.8570065791964926.07120335228367.132347149
1965020.79586278228396.9247803571965236.98198067228124.209430223
#Sta/Elev= 30
       0 1914.62    11.1 1910.24    45.5 1909.48    55.8 1907.82    65.3 1903.09
    76.5 1895.77      94 1889.99  114.691885.738   128.9 1883.65   156.5  1884.3
  162.271885.738   180.5 1890.26   206.1 1892.98     213 1895.55   234.1 1899.42
     287 1897.91   301.8 1899.78   313.5 1903.65   321.9 1909.36   339.9 1924.81
   355.4 1927.89   357.9 1929.38   369.5 1940.35   418.2 1972.71   443.3 1991.14
     460 2004.95   493.5 2028.84   523.7 2048.45     533  2055.7   546.6  2061.8
#Mann= 6 ,-1 , 0
       0      .1       0      50     .04       0  114.69    .045       0
  162.27     .04       0   308.6      .1       0   428.6     .12       0
#XS Ineff= 2 , 0
           111.5 1885.93  165.97         1886.02
Permanent Ineff=
       F       F
Bank Sta=114.69,162.27
XS Rating Curve= 0 ,0
Exp/Cntr(USF)=0,0
Exp/Cntr=0.5,0.3

Type RM Length L Ch R = 1 ,32029   ,160.7,160.4,159.6
XS GIS Cut Line= 4
1964903.36544458 228585.435639081964933.53370117228539.295952532
1965063.07974417228393.7784795731965238.76547372228163.080046834
#Sta/Elev= 30
       0 1968.34      31 1950.17    50.8 1936.72    67.2 1929.65    97.4 1910.54
   106.2 1906.26   111.1 1899.17  118.441883.985   120.6 1880.76     123 1880.56
  152.19 1883.98     181    1888   206.6 1889.71   221.4 1895.09   236.8  1895.1
   268.5 1898.09   287.1 1898.27   297.9 1896.72   313.8 1897.63   326.2 1900.09
   330.4 1902.31   346.8 1916.45   350.9 1918.88   368.3 1922.79   372.5 1926.63
   379.8 1935.69     410 1954.65   441.7 1976.58     482 2009.28   539.9 2046.32
#Mann= 6 ,-1 , 0
       0      .1       0  118.44    .045       0  152.19      .1       0
  225.13     .04       0  349.95      .1       0  479.95     .12       0
Bank Sta=118.44,152.19
XS Rating Curve= 0 ,0
Exp/Cntr(USF)=0,0
Exp/Cntr=0.3,0.1

Type RM Length L Ch R = 1 ,31869   ,210.4,206.1,202.8
XS GIS Cut Line= 4
1964965.47656109228750.4737486561965047.10831421228656.419772231
1965190.85118384228484.2832493411965403.80358329228372.483239628
#Sta/Elev= 30
       0 1990.76    35.7 1972.24   139.7 1907.69   153.1 1901.21     161 1899.46
   178.7 1891.22   188.1  1888.4     195 1883.59  201.281880.839   225.2 1878.77
  244.92 1880.84   246.5  1881.6   253.3 1889.47   259.4 1891.81   276.5 1891.84
   292.9 1893.57   365.8 1894.36   370.7 1895.56   384.6 1904.65   404.1 1920.82
   409.5 1926.36   415.2 1935.54   418.9 1938.71   441.2 1951.25   482.4 1978.96
   496.7 1986.48     514 1993.17     531  2002.6   560.2 2011.32   589.3 2021.77
#Mann= 6 ,-1 , 0
       0      .1       0  201.28    .045       0  244.92      .1       0
  314.54     .04       0   418.8     .12       0   498.8      .1       0
Bank Sta=201.28,244.92
XS Rating Curve= 0 ,0
Exp/Cntr(USF)=0,0
Exp/Cntr=0.3,0.1

Type RM Length L Ch R = 1 ,31663   ,279.2,274.6,268.5
XS GIS Cut Line= 4
1965091.47339743228897.7658249431965196.17499383228796.613435204
1965307.97500354228628.0261189711965457.04168315228452.340389423
#Sta/Elev= 30
       0 1975.23    14.6 1967.94    42.5 1956.82    87.6 1933.77   145.6 1896.71
     154 1892.49   162.4 1889.97   170.3 1881.07   177.41877.104   182.1 1875.29
   200.7 1874.09   212.6 1874.31  222.461877.104   232.1 1879.52     249 1878.26
   256.9 1882.59   260.8 1883.46   300.2 1885.79   319.9 1884.66   326.8 1886.05
   347.9 1901.84   377.5 1932.18   389.5 1942.33   424.9 1968.17     442 1978.94
   459.8 1988.59   487.8 1998.46   504.1 2005.97   548.3 2017.68   578.3 2027.96
#Mann= 6 ,-1 , 0
       0      .1       0   177.4    .045       0  222.46      .1       0
  255.58     .12       0  507.87      .1       0  567.87     .12       0
#XS Ineff= 2 , 0
                          233.81         1888.03
Permanent Ineff=
       F       F
Bank Sta=177.4,222.46
XS Rating Curve= 0 ,0
Exp/Cntr(USF)=0,0
Exp/Cntr=0.3,0.1

Type RM Length L Ch R = 1 ,31388   ,240.3,232.4,215.8
XS GIS Cut Line= 4
1965288.45436692229092.9721911081965396.70516998 228931.48328819
 1965490.7591464228775.3181952581965556.41946957228500.254679299
#Sta/Elev= 30
       0 1989.59    49.8 1958.23     109 1919.03   141.3 1900.25   155.5 1892.91
   168.3 1887.77   180.1 1884.16   195.7 1881.68     238 1879.38   250.7 1874.55
   268.6 1871.94   286.6 1872.26   291.6 1874.28   314.6 1873.84   318.4 1873.13
   326.1 1870.75     332 1871.38  335.831873.313   337.6 1875.04   348.7 1892.46
   352.9  1897.1   364.4 1907.09   415.6 1937.45   443.4 1949.53   578.4 1987.81
   591.9 1992.96   606.2 1999.53   636.2 2014.93   649.2 2023.05   659.5 2028.54
#Mann= 8 ,-1 , 0
       0     .08       0     110      .1       0  294.41     .12       0
   318.4    .045       0  335.83     .12       0  446.72      .1       0
  546.72     .12       0  606.72      .1       0
Bank Sta=318.4,335.83
XS Rating Curve= 0 ,0
Exp/Cntr(USF)=0,0
Exp/Cntr=0.3,0.1

Type RM Length L Ch R = 1 ,31156   ,207.9,200.9,187.7
XS GIS Cut Line= 4
1965488.98454307229259.7849040121965575.94010618229084.099174464
1965662.89566929228832.1055017791965701.93694252228473.635629368
#Sta/Elev= 30
       0 2025.37    50.2 1992.06   162.8 1907.04   188.3 1891.21   209.6 1883.12
   233.9 1879.43   244.3 1879.81   254.7 1875.05  273.431869.104   279.7 1866.88
   289.4 1866.35   310.7 1867.74   315.81869.109   324.1 1873.01   341.4 1875.89
   355.3  1877.6   379.6 1878.08   393.5 1887.48   410.9 1905.75   459.4 1927.96
   575.1 1947.17   633.2 1962.12   690.6 1978.94   713.7 1984.64   723.6 1985.94
   739.8 1991.11   753.3 1995.94   796.3 2015.89   809.4 2025.23   823.2 2036.83
#Mann= 5 ,-1 , 0
       0      .1       0  273.43    .045       0   315.8      .1       0
  386.03     .12       0   692.6      .1       0
Bank Sta=273.43,315.8
XS Rating Curve= 0 ,0
Exp/Cntr(USF)=0,0
Exp/Cntr=0.3,0.1

Type RM Length L Ch R = 1 ,30955   ,232.9,230.9,225.6
XS GIS Cut Line= 4
1965817.28615889 229348.515070451965803.08933226229098.296001094
1965801.31472894228842.7531217511965755.17504239228454.114992752
#Sta/Elev= 30
       0 1999.72    41.1 1973.88    67.3 1953.52   126.5 1911.69   146.2 1899.56
   172.3 1886.91   198.8 1882.73   231.6 1881.78   274.3 1878.79     294 1875.09
   313.7 1874.97   323.5 1865.88   330.1 1863.65   349.8 1863.85  359.691865.881
   366.2 1868.09   412.1 1870.69   427.5  1881.1   444.9 1898.11   458.1 1905.08
     481 1913.46   540.3 1929.69   553.5 1931.18   665.9 1958.93   715.4 1975.32
     735  1978.2   814.5  2000.1     841 2012.59   877.3 2038.39   897.5  2050.3
#Mann= 5 ,-1 , 0
       0      .1       0   323.5    .045       0  359.69      .1       0
  450.62     .12       0  746.17      .1       0
#XS Ineff= 2 , 0
                          378.22         1882.35
Permanent Ineff=
       F       F
Bank Sta=323.5,359.69
XS Rating Curve= 0 ,0
Exp/Cntr(USF)=0,0
Exp/Cntr=0.3,0.1

Type RM Length L Ch R = 1 ,30724   ,317.5,325.6,334.3
XS GIS Cut Line= 4
1966058.63221161229394.6547569981966040.88617832229073.451554491
1966003.61950841228791.2896252171965977.00045848228392.003876245
#Sta/Elev= 30
       0  1962.5      61 1935.76   126.7  1899.2   169.4 1881.81   189.1 1876.19
   235.1 1871.65   342.6  1870.3   386.7 1863.77   403.3 1864.95  413.451861.877
   429.8 1859.37     443 1859.55  446.631861.874   462.8 1879.66     479 1892.38
   495.9  1904.2   512.5 1912.62   621.6 1944.31     654    1950   687.4 1951.92
   726.8 1962.16   756.4 1971.96   772.8 1979.01   799.2 1993.96   832.8 2005.45
   845.2 2011.84   882.1 2035.84     934 2064.11   966.8 2084.79  1006.5 2113.86
#Mann= 6 ,-1 , 0
       0      .1       0  391.69     .12       0  413.45    .045       0
  446.63     .12       0  591.69      .1       0  986.31     .12       0
#XS Ineff= 2 , 0
          398.85 1875.66
Permanent Ineff=
       F       F
Bank Sta=413.45,446.63
XS Rating Curve= 0 ,0
Exp/Cntr(USF)=0,0
Exp/Cntr=0.3,0.1

Type RM Length L Ch R = 1 ,30398   ,307.5,303.9,284.9
XS GIS Cut Line= 4
 1966305.3020743229415.9499969431966328.37191758229085.873777792
1966365.63858748228839.203915094 1966385.1592241228459.438802738
#Sta/Elev= 30
       0 1933.78   121.8 1887.49   148.2 1876.03   177.8 1868.48   263.3  1863.7
   309.3 1863.31   332.3 1859.96   365.5    1861   385.4  1858.4   405.3 1859.69
   415.3 1857.29     425 1857.16   441.8 1854.55  470.961857.334     475    1860
   488.3  1874.1   498.2 1879.81   561.3 1902.99   587.8    1917     613  1932.8
   643.6 1958.72   666.6 1973.08   679.7 1984.42   725.7  2017.8   768.8 2042.01
   786.1 2053.82     815 2068.59   880.1 2110.89     936 2139.49   960.6  2153.7
#Mann= 6 ,-1 , 0
       0      .1       0  420.88     .12       0     425    .045       0
  470.96     .12       0  620.35      .1       0  710.35     .12       0
#XS Ineff= 2 , 0
          405.44 1872.26
Permanent Ineff=
       F       F
Bank Sta=425,470.96
XS Rating Curve= 0 ,0
Exp/Cntr(USF)=0,0
Exp/Cntr=0.3,0.1

Type RM Length L Ch R = 1 ,30094   ,227.2,220,208.4
XS GIS Cut Line= 4
1966676.19417002229399.9785669841966649.57512009229156.857910943
1966587.46400358228895.9912216141966450.81954726228454.114992752
#Sta/Elev= 30
       0 1970.34    76.5 1941.47   110.1 1934.63   182.1  1915.5   288.7 1870.24
   305.5 1860.46   317.5 1858.54  330.721851.547   339.3 1848.94  372.871851.548
   386.5 1854.58   511.3 1855.23   521.5 1855.94   529.4 1859.44   558.2 1881.28
   571.3 1886.87   590.2 1902.42   615.9 1920.24   631.4 1934.13   645.9 1945.28
   676.1 1964.35   699.8 1982.23   723.5 1995.05   751.6 2013.52   786.4 2039.74
   844.3 2074.73     889 2094.93   914.9 2110.13   930.7 2116.02   975.3 2139.84
#Mann= 4 ,-1 , 0
       0      .1       0  330.72    .045       0  372.87     .12       0
  812.73      .1       0
#XS Ineff= 2 , 0
                          388.25         1869.08
Permanent Ineff=
       F       F
Bank Sta=330.72,372.87
XS Rating Curve= 0 ,0
Exp/Cntr(USF)=0,0
Exp/Cntr=0.3,0.1

Type RM Length L Ch R = 1 ,29874   ,371.6,370.4,362.9
XS GIS Cut Line= 4
1966997.39737252 229261.55950734 1966890.9211728229073.451554491
1966715.23544325228785.9658152311966493.41002715228447.016579436
#Sta/Elev= 30
       0 2058.51    82.9 2005.24   154.5 1953.69   241.7 1894.71   253.3 1881.64
   268.5 1879.45   280.4 1869.73   304.3 1854.58  344.59 1847.28   349.6 1845.76
   373.5 1845.46  402.341847.279   411.7 1849.04   442.7 1847.58   457.1 1849.66
   482.1 1848.89   503.2 1852.41   579.3 1880.99   608.1 1893.84     663 1926.47
   719.1 1966.09   730.2 1970.24   745.3 1981.45   757.1 1987.05   764.9 1993.23
   772.8 1996.54   803.7 2016.34   843.3  2036.6   917.8 2098.18   958.2 2125.67
#Mann= 5 ,-1 , 0
       0      .1       0  296.15     .04       0  344.59    .045       0
  402.34     .12       0  536.15      .1       0
#XS Ineff= 2 , 0
                          415.47          1861.4
Permanent Ineff=
       F       F
Bank Sta=344.59,402.34
XS Rating Curve= 0 ,0
Exp/Cntr(USF)=0,0
Exp/Cntr=0.3,0.1

Type RM Length L Ch R = 1 ,29504   ,452.8,469.7,494
XS GIS Cut Line= 4
1967235.19421858229128.4642576831967153.56246546228929.708684861
  1966940.610066228551.7181758341966686.84178999228219.867353354
#Sta/Elev= 30
       0 2074.11    22.8 2064.47   132.7 1979.05   157.6 1962.14   182.4 1940.85
   241.7 1882.13     282 1848.36   300.9 1842.38   407.9 1844.93   441.7  1844.1
  449.36 1840.94   470.6 1838.35   485.4 1840.51     508 1843.23   523.6 1841.65
     538 1849.47   553.2 1863.88   562.1 1869.58   663.7 1902.55   747.1 1939.31
   803.3 1973.08   845.4 2002.57   861.6 2010.91   899.2  2037.7   915.6    2046
   940.4 2063.66   961.1 2075.28     975 2078.99  1039.7 2113.13  1066.5 2129.52
#Mann= 5 ,-1 , 0
       0      .1       0  354.87     .12       0  449.36    .045       0
   485.4     .12       0  688.72      .1       0
#XS Ineff= 2 , 0
           429.8 1853.73
Permanent Ineff=
       F       F
Bank Sta=449.36,485.4
XS Rating Curve= 0 ,0
Exp/Cntr(USF)=0,0
Exp/Cntr=0.3,0.1

Type RM Length L Ch R = 1 ,29034   ,407.7,417.6,425
XS GIS Cut Line= 4
1967352.31803828229080.5499678061967398.45772483228867.597568354
1967455.24503135 228643.997548931967650.45139751228086.772103697
#Sta/Elev= 30
       0 2041.19    22.9 2027.29    96.7 1970.99   123.6 1952.88   244.7 1857.15
   267.2 1837.53   275.1 1834.06   312.4 1834.76  321.181833.022   325.9 1830.92
   332.7 1830.55   356.4 1831.01  361.26    1833   366.5 1837.43   373.3 1837.89
   403.8 1837.53   418.3 1835.23   470.4 1835.68   520.7 1832.88   548.6 1834.09
   614.6 1864.02   635.5 1875.76   680.7 1884.93   722.4 1904.64   830.1 1980.61
   856.6 1995.98   889.2 2017.91   935.7 2046.57  1003.3 2092.58    1039 2110.51
#Mann= 6 ,-1 , 0
       0      .1       0  321.18    .045       0  361.26      .1       0
  387.89     .12       0  588.59      .1       0  928.59     .12       0
#XS Ineff= 2 , 0
          287.06 1838.28  381.66         1850.66
Permanent Ineff=
       F       F
Bank Sta=321.18,361.26
XS Rating Curve= 0 ,0
Exp/Cntr(USF)=0,0
Exp/Cntr=0.3,0.1

Type RM Length L Ch R = 1 ,28617   ,231.3,225.1,219.5
XS GIS Cut Line= 4
1967636.25457088229169.2801342451967710.78791069 228988.27059471
1967870.50221028 228672.39120219 1967964.5561867228310.372123121
#Sta/Elev= 30
       0 1960.23    20.8 1948.47    76.4 1913.39     113 1892.51   173.4 1862.44
     202 1855.74   216.6 1849.51   231.8 1840.05   243.4 1834.63   257.1 1830.59
   275.5 1828.24   315.9 1828.73   345.3 1830.51   385.8 1829.92  427.981824.233
     452 1822.48     473 1822.58  478.231824.238   481.4 1827.63   492.4 1849.06
   496.1 1854.65     507 1862.41   521.8 1875.45   547.5 1893.05   679.9 1967.95
   734.1 2004.36   798.6 2040.52     866 2084.52   895.6  2099.1   923.8 2109.62
#Mann= 6 ,-1 , 0
       0      .1       0  405.75     .12       0  427.98    .045       0
  478.23     .12       0  619.72      .1       0  699.72     .12       0
#XS Ineff= 2 , 0
          369.63 1845.29
Permanent Ineff=
       F       F
Bank Sta=427.98,478.23
XS Rating Curve= 0 ,0
Exp/Cntr(USF)=0,0
Exp/Cntr=0.3,0.1

Type RM Length L Ch R = 1 ,28392   ,241.7,221.1,188.4
XS GIS Cut Line= 4
1967854.53078032229227.8420440941967920.19110348229052.156314546
1967998.27364995 228787.740418561968014.24507991228344.089586368
#Sta/Elev= 30
       0 1914.39      41  1891.9      62 1882.14      86 1872.28   181.1 1838.76
   212.1  1826.1   222.3 1824.09   283.9 1824.43  297.181819.865   312.1 1816.56
     342 1819.44   383.1 1820.23     407 1825.45   437.8 1860.91   465.1 1884.86
   503.8  1912.8   507.8 1916.39   514.4 1925.12   520.9 1930.49   576.7 1969.19
   589.9 1976.97   645.7 2005.35   671.9 2016.62   708.1 2029.59   734.3 2041.27
   741.4 2048.34   809.8 2083.68   842.7 2095.47   865.6 2102.11   907.2 2108.39
#Mann= 5 ,-1 , 0
       0      .1       0  297.18    .045       0     342      .1       0
  347.55     .12       0  743.26      .1       0
Bank Sta=297.18,342
XS Rating Curve= 0 ,0
Exp/Cntr(USF)=0,0
Exp/Cntr=0.3,0.1

Type RM Length L Ch R = 1 ,28171   ,262,271.9,252.3
XS GIS Cut Line= 6
1967912.23088622229133.7081836691968070.08419262229096.522799662
1968193.48001611229071.6769511621968097.65143636228892.442014957
1968071.03238643228810.8102618341968053.28635314228358.286412998
#Sta/Elev= 30
       0 1861.13    72.3 1836.86    99.2 1829.64   223.5 1827.12     267 1822.86
   325.7 1822.77   342.3 1820.91     348 1816.83   364.2 1814.66   396.4 1816.46
   415.1 1817.08   436.9 1820.72     464 1819.51   505.8 1821.17   527.5 1818.57
   534.5 1819.52   544.6  1826.1   573.4 1858.55   595.5 1878.35   644.8 1914.05
   661.3 1928.39   727.4  1971.1   795.8 2009.88   871.3 2044.97     880  2053.1
     914 2069.64   930.4 2083.67   945.4 2091.34   976.4 2103.03    1030 2108.28
#Mann= 6 ,-1 , 0
       0      .1       0 215.607     .12       0 239.354      .1       0
     348    .045       0   396.4     .12       0 863.845      .1       0
#XS Ineff= 2 ,-1
       0   300.4 1832.95  416.071003.572  1832.4
Permanent Ineff=
       F       F
Bank Sta=348,396.4
XS Rating Curve= 0 ,0
Exp/Cntr(USF)=0,0
Exp/Cntr=0.3,0.1

Type RM Length L Ch R = 1 ,27899   ,340.4,321.5,311.1
XS GIS Cut Line= 4
1968608.73719504229183.476960875 1968340.7720924228883.568998313
1968197.02922277228674.1658055191968078.13079974228360.061016327
#Sta/Elev= 30
       0 1932.73    44.8 1913.84   132.8 1868.92   176.6 1852.63   207.6 1838.76
   234.8 1817.31   299.9 1818.13   304.4 1817.94   309.5 1814.93   348.6 1817.71
     409 1815.67   429.1  1816.9   501.2 1815.33  509.041812.726   536.6 1810.06
     546 1810.44  551.171812.726   579.1 1826.19   636.1 1865.62   659.5 1884.71
   691.1 1903.74   705.1 1910.52   750.7 1943.65   848.9 2006.98   866.5 2022.44
   903.8 2046.08   912.1 2056.34   937.6 2077.37   957.7 2088.32     992  2097.3
#Mann= 8 ,-1 , 0
       0     .12       0     380      .1       0  482.18     .12       0
  502.18      .1       0  509.04    .045       0  551.17      .1       0
  726.17     .12       0  836.17      .1       0
#XS Ineff= 2 , 0
          432.39 1817.94
Permanent Ineff=
       F       F
Bank Sta=509.04,551.17
XS Rating Curve= 0 ,0
Exp/Cntr(USF)=0,0
Exp/Cntr=0.3,0.1

Type RM Length L Ch R = 1 ,27577   ,275.6,269.9,267.5
XS GIS Cut Line= 4
1968840.58948509228739.7336253541968660.45142428228618.018719403
1968353.72986129228471.9608322621968127.34013622228333.205839478
#Sta/Elev= 30
       0  1974.1   138.1 1885.44     183  1859.9   206.7 1849.32   255.5 1834.75
   274.2 1825.19   292.3 1813.16   303.2 1807.65     325 1803.48     365 1807.76
     405 1806.15   426.8 1805.01   442.5 1806.26   467.2 1807.57   484.9 1813.38
   532.2 1838.96   550.9 1851.02     578 1869.42   623.1 1903.84   669.2 1943.18
     691 1958.99     700 1970.78   709.8 1976.78   726.9 1991.91   738.5 1998.53
   751.4 2009.87   761.6 2015.16   803.8 2042.55   815.5 2056.39   822.7 2061.07
#Mann= 7 ,-1 , 0
       0      .1       0      60     .12       0     180      .1       0
   297.4     .12       0     405    .045       0   442.5     .12       0
  627.13      .1       0
#XS Ineff= 2 , 0
          365.06 1811.84
Permanent Ineff=
       F       F
Bank Sta=405,442.5
XS Rating Curve= 0 ,0
Exp/Cntr(USF)=0,0
Exp/Cntr=0.3,0.1

Type RM Length L Ch R = 1 ,27307   ,301.6,301.1,299.1
XS GIS Cut Line= 4
1969035.33333461228479.2637266191968772.42913776228350.245926311
1968460.83897852228240.702510955 1968227.1463591228131.159095599
#Sta/Elev= 30
       0 2096.83    32.5 2070.91    56.2 2057.98    98.3 2028.84   193.3 1956.63
   240.8 1927.51   265.8 1906.57   316.3 1868.94   340.7 1847.31   396.3 1821.31
   403.3 1814.95   413.7 1802.09     452 1798.61   476.3 1799.14   500.7 1804.66
     518 1802.78     532 1804.57   542.3 1801.06   556.3 1800.94   566.7 1803.87
   591.3  1805.9   629.6 1836.64   680.3  1866.2   755.4 1905.89   791.9 1929.11
   807.3 1943.01   822.8 1952.56   856.5 1977.99   868.7 1984.77   881.2 1995.14
#Mann= 5 ,-1 , 0
       0      .1       0  402.86     .12       0  482.86      .1       0
   542.3    .045       0   556.3      .1       0
#XS Ineff= 2 , 0
          499.04 1808.89
Permanent Ineff=
       F       F
Bank Sta=542.3,556.3
XS Rating Curve= 0 ,0
Exp/Cntr(USF)=0,0
Exp/Cntr=0.3,0.1

Type RM Length L Ch R = 1 ,27006   ,306.4,312.4,315.8
XS GIS Cut Line= 4
1969093.75648947228274.7826846211968857.62957193  228080.0388351
1968514.39353714227960.758227267  1968266.095129227924.243755482
#Sta/Elev= 30
       0 2085.87    11.4 2080.78    15.7 2076.39    32.7  2051.6    44.1 2046.09
    52.7 2038.28    74.4 2026.52   150.7 1978.82   186.8  1953.3   219.8 1927.48
     295 1875.74   377.2 1828.66   423.2 1797.12     444 1795.07   482.2 1796.14
   489.2 1794.87   499.6 1794.91  504.81 1796.72     510 1799.47   520.5 1800.74
     576 1800.23   606.6 1802.26   669.8 1835.01   696.3 1856.72   706.3 1862.49
   782.5 1926.57     810  1950.6   838.6 1980.11   898.6 2030.76   920.4 2051.37
#Mann= 4 ,-1 , 0
       0      .1       0  376.07     .12       0   482.2    .045       0
  504.81      .1       0
#XS Ineff= 2 , 0
                          526.45         1802.76
Permanent Ineff=
       F       F
Bank Sta=482.2,504.81
XS Rating Curve= 0 ,0
Exp/Cntr(USF)=0,0
Exp/Cntr=0.3,0.1

Type RM Length L Ch R = 1 ,26694   ,295.8,294.1,293.5
XS GIS Cut Line= 4
1969183.82551987227987.5355065771968957.43579481227824.437532602
1968699.40019419 227680.813943581968460.83897852227566.401931986
#Sta/Elev= 30
       0 2034.39    71.1 1986.63   109.8 1962.21   170.4  1919.8   213.4 1890.98
   255.7 1865.45   290.8 1847.65   303.4 1843.21   335.9 1828.82   351.6 1820.11
   388.4 1797.04   407.2 1792.56     441 1791.83   452.3  1789.7   467.6 1789.56
   478.6 1790.31   481.9 1791.97   489.8 1795.65   515.6 1795.91   548.5 1801.32
   568.8 1803.42   590.7 1809.35     635  1816.6   656.2 1824.14   681.7 1839.54
   707.1  1858.9   772.9 1912.08   787.2 1921.68   814.5  1943.2   838.9 1957.61
#Mann= 3 ,-1 , 0
       0      .1       0     441    .045       0   481.9      .1       0
Bank Sta=441,481.9
XS Rating Curve= 0 ,0
Exp/Cntr(USF)=0,0
Exp/Cntr=0.3,0.1

Type RM Length L Ch R = 1 ,26400   ,326.9,324.7,329.3
XS GIS Cut Line= 4
1969337.18630137227675.9453473421969101.05938383227563.967633867
1968704.26879043227366.7894862261968524.13072962227301.063437013
#Sta/Elev= 30
       0 2002.14    16.2 1990.75    35.9 1979.81   104.9 1932.74   181.2 1884.58
   195.7  1877.9   224.7 1861.35   265.5 1841.96   301.7 1820.88   340.8 1796.06
   360.4 1788.99   378.3  1788.8   403.9 1791.25   411.2 1788.83   418.6 1786.66
   441.2 1786.56   450.41788.085   465.6 1788.97   502.8 1787.53   561.5  1791.4
   572.4 1795.87   598.9 1810.74   627.2 1820.12   663.9 1835.31   704.4 1863.16
   734.7 1888.35   742.8 1893.69   798.6 1945.05   826.6  1966.8   896.2  2025.7
#Mann= 3 ,-1 , 0
       0      .1       0   411.2    .045       0   450.4      .1       0
#XS Ineff= 2 , 0
          402.64 1795.86
Permanent Ineff=
       F       F
Bank Sta=411.2,450.4
XS Rating Curve= 0 ,0
Exp/Cntr(USF)=0,0
Exp/Cntr=0.3,0.1

Type RM Length L Ch R = 1 ,26075   ,618.7,630.9,632.8
XS GIS Cut Line= 4
1969434.55822613227459.2928147491969230.07718414 227308.36633137
1968830.85229262227103.8852893721968604.46256755226977.301787183
#Sta/Elev= 30
       0 1971.84     5.2 1969.02    21.6 1956.04    79.8 1913.43      92 1906.06
   129.6 1879.89   148.3 1864.09   185.9 1839.11   224.6 1820.72   254.1 1808.52
   291.9  1794.7   317.7 1788.51   347.2 1785.62   409.7 1786.81   472.5 1786.49
   498.3 1784.16   549.9 1784.06   572.1 1781.53   586.8  1782.4   591.1 1784.13
     600  1794.1   616.3  1808.9     631 1819.85   645.8 1827.04   707.2 1851.93
   738.8 1866.66   785.6 1892.22   861.5    1938   899.9 1958.73   962.1 1995.71
#Mann= 5 ,-1 , 0
       0      .1       0     220     .12       0  304.15      .1       0
   549.9    .045       0   591.1      .1       0
#XS Ineff= 2 , 0
          477.08 1804.28
Permanent Ineff=
       F       F
Bank Sta=549.9,591.1
XS Rating Curve= 0 ,0
Exp/Cntr(USF)=0,0
Exp/Cntr=0.3,0.1

Type RM Length L Ch R = 1 ,25444   ,312.1,311.8,314.6
XS GIS Cut Line= 4
1969653.64505685227164.7427423471969461.33550544226982.170383421
1969232.51148225226789.8608320181969003.68745907226595.116982496
#Sta/Elev= 30
       0 1991.41    28.4 1974.08   128.2 1903.45   141.8 1892.28   150.9 1887.35
   160.6 1878.15   169.9 1871.55   194.8 1858.55   256.7  1822.3   269.7 1808.17
   281.2 1804.02   285.4  1800.8   298.3 1777.62  304.631773.771     314 1771.57
   337.3 1771.93   345.4 1774.07     354 1774.57   374.5 1771.92   386.1    1776
   397.8 1777.84   511.1 1776.75   521.3 1777.76   529.7 1780.68   577.3  1818.9
   624.3 1860.59   642.3  1870.3   665.5 1889.55   735.4 1940.54   864.6 2042.59
#Mann= 5 ,-1 , 0
       0     .12       0      50      .1       0  304.63    .045       0
   345.4     .04       0  375.17      .1       0
Bank Sta=304.63,345.4
XS Rating Curve= 0 ,0
Exp/Cntr(USF)=0,0
Exp/Cntr=0.3,0.1

Type RM Length L Ch R = 1 ,25132   ,265.6,271.9,284.7
XS GIS Cut Line= 4
1969807.00583834226991.9075758971969636.60497001226748.477763995
1969446.72971673226565.9054050681969045.07052709226451.493393474
#Sta/Elev= 30
       0 1979.11    80.9 1917.96   118.5 1894.95     145 1876.08     165 1865.04
   206.5 1838.67   238.6 1816.37   325.5 1775.91     3871765.384     398 1764.04
   424.9 1766.18   443.7 1764.01   457.6 1768.88   493.6  1770.4   514.9 1778.03
   548.1  1781.5   585.4 1782.53   602.1 1785.39   617.5 1790.27   663.8 1812.45
   701.4 1833.72   735.5 1856.15   766.2 1873.81   820.8 1911.31   827.6 1914.76
   886.1 1955.49   906.1  1967.3   919.7 1979.45   933.3 1988.91   978.2 2009.49
#Mann= 3 ,-1 , 0
       0      .1       0     387    .045       0   424.9      .1       0
#XS Ineff= 2 , 0
                          465.62         1788.16
Permanent Ineff=
       F       F
Bank Sta=387,424.9
XS Rating Curve= 0 ,0
Exp/Cntr(USF)=0,0
Exp/Cntr=0.3,0.1

Type RM Length L Ch R = 1 ,24860   ,347.3,380.4,390
XS GIS Cut Line= 4
1969982.27530291226938.3530172781969867.86329132226699.791801614
 1969712.0682117226380.8987480221969522.19295842226008.451135812
#Sta/Elev= 30
       0 2004.73   126.9  1912.3   163.3 1883.49   214.2 1848.61   232.4 1837.75
   261.5 1816.01   316.3 1779.07   335.2 1770.75   363.8  1766.5   378.4  1761.2
   389.2 1761.34   396.4 1759.29   407.6 1758.64   426.3  1759.6  433.991761.451
   448.1 1766.09   558.5 1769.93   568.3  1773.2   579.2  1779.2     623 1794.26
   688.1 1820.77   708.2 1829.15   744.2 1846.59   822.9 1895.29     859 1921.21
     881 1938.35   960.1 2004.87   987.6 2023.85  1019.8 2051.04  1037.5 2063.72
#Mann= 6 ,-1 , 0
       0      .1       0   389.2    .045       0  433.99      .1       0
  699.49     .12       0  769.49      .1       0  919.49     .12       0
Bank Sta=389.2,433.99
XS Rating Curve= 0 ,0
Exp/Cntr(USF)=0,0
Exp/Cntr=0.3,0.1

Type RM Length L Ch R = 1 ,24480   ,367.2,407.7,426.3
XS GIS Cut Line= 4
1970089.38442015 226933.484421041970125.89889194226558.602510711
1970152.67617124226329.7784875231970213.53362422 225838.05026748
#Sta/Elev= 30
       0 1995.93   114.8  1911.5     176 1864.82     217 1836.44     271 1796.46
   281.5 1790.48   324.3 1773.47     354 1764.21   380.4 1761.54   426.4 1761.76
   439.8 1757.73   453.1 1756.81  469.151752.598   485.6 1750.31   512.5 1751.09
  520.361752.598   525.7 1755.94   548.8 1776.92   558.7 1782.82     607 1797.25
   697.6 1830.22   730.4 1839.94   790.1 1861.64   826.5 1877.24   868.6  1899.5
   906.9  1917.5   938.9 1935.44   983.4 1963.46  1011.6 1982.81  1102.5 2037.71
#Mann= 5 ,-1 , 0
       0      .1       0  469.15    .045       0  520.36      .1       0
  787.04     .12       0  987.04      .1       0
Bank Sta=469.15,520.36
XS Rating Curve= 0 ,0
Exp/Cntr(USF)=0,0
Exp/Cntr=0.3,0.1

Type RM Length L Ch R = 1 ,24072   ,404.6,413.5,406.8
XS GIS Cut Line= 4
1970167.28195996226943.2216135161970310.90554898226772.820745185
1970680.91886307226473.4020765451971036.32638845226166.680513548
#Sta/Elev= 30
       0 1973.11   138.8 1860.87     186 1827.69   233.9 1799.38   278.2  1765.1
   287.6 1760.58   301.6 1757.34   312.8  1748.4  357.621744.068   376.1 1741.19
   401.9 1741.64  416.191744.067   488.2 1785.09   509.2 1794.79   527.8 1798.88
   564.1  1801.1   582.9 1804.67     604 1811.62   722.8 1840.96   757.5 1853.24
     795 1863.33   812.1 1870.38   830.2 1880.68   852.9 1899.06   870.4 1909.77
   886.5 1924.74   991.2  2012.1  1009.8 2026.04    1061 2062.55  1168.3 2132.41
#Mann= 8 ,-1 , 0
       0     .08       0      10      .1       0  357.62    .045       0
  416.19      .1       0  422.85     .12       0  432.85      .1       0
  682.85     .12       0  808.84      .1       0
Bank Sta=357.62,416.19
XS Rating Curve= 0 ,0
Exp/Cntr(USF)=0,0
Exp/Cntr=0.3,0.1

Type RM Length L Ch R = 1 ,23659   ,373.4,385.6,387
XS GIS Cut Line= 4
1970400.97457939227184.217127299 1970517.8208891227089.279500658
1970729.60482545226904.272843612  1971170.212785226638.934348639
#Sta/Elev= 30
       0  1867.3    54.4 1845.64    82.3 1831.83   104.2 1822.83   208.3  1769.4
     216 1764.17   225.7 1754.82   238.8 1746.61   249.7 1745.23   269.4 1739.24
   282.3 1737.56   306.6 1738.77   334.5 1739.34   348.5 1745.53   364.4 1746.93
   382.5 1744.78     413  1744.3   453.7 1744.46     473 1746.06   487.2 1750.43
     511 1763.78   525.4 1770.12   572.3 1782.31   599.1 1793.81   671.9 1841.85
   740.8 1894.95   775.3 1916.49   800.3 1935.29     829 1954.02   946.1 2039.21
#Mann= 5 ,-1 , 0
       0      .1       0   269.4    .045       0   306.6      .1       0
  380.55     .12       0  471.76      .1       0
Bank Sta=269.4,306.6
XS Rating Curve= 0 ,0
Exp/Cntr(USF)=0,0
Exp/Cntr=0.3,0.1

Type RM Length L Ch R = 1 ,23273   ,458.3,464,452.5
XS GIS Cut Line= 4
1970493.47790791227437.3841316781970702.82754614 227308.36633137
1970936.52016557227206.1258103711971206.72725678 227108.75388561
#Sta/Elev= 30
       0 1874.83    75.8 1832.38   125.9 1808.01   160.6 1788.49     176 1777.86
   199.1 1757.33   231.2 1738.08   244.8 1735.98     360 1737.35   374.2 1734.76
   406.41733.484   420.9 1730.57   431.6 1730.59   435.2 1731.39  436.88 1733.48
   449.5 1751.43   467.4 1766.92   478.2 1780.71   488.6 1789.95   510.2 1803.12
   524.1  1815.9   579.9 1845.22   611.3 1863.53     688 1912.39   712.4 1930.32
   726.4 1938.62   747.3 1948.85   764.7 1955.18   778.7 1958.63   788.2 1958.35
#Mann= 5 ,-1 , 0
       0      .1       0   406.4    .045       0  436.88     .12       0
  630.99      .1       0  740.99     .12       0
#XS Ineff= 2 , 0
          359.89 1753.29
Permanent Ineff=
       F       F
Bank Sta=406.4,436.88
XS Rating Curve= 0 ,0
Exp/Cntr(USF)=0,0
Exp/Cntr=0.3,0.1

Type RM Length L Ch R = 1 ,22809   ,288.5,280.6,268.4
XS GIS Cut Line= 4
1970471.56922484227766.0143777461970646.83868941227702.722626651
1970895.13709755227627.2593849611971175.08138123227529.887460201
#Sta/Elev= 30
       0 1889.41    32.6 1870.38    67.5 1857.18   116.3 1836.15   144.2 1821.07
   162.7 1807.94   210.1 1787.86   230.7 1777.19   234.1 1774.75     236 1771.48
   244.4 1751.15   247.8 1744.66   261.5 1733.32   275.4 1725.53     289  1723.7
   326.7 1725.94   357.5 1729.58   429.6 1733.09   443.3 1736.93   451.3 1741.75
     471 1757.34   490.6 1769.99   554.4 1817.79   589.1 1837.28   606.5 1845.23
   658.6 1874.73   686.4 1888.38   710.7 1899.32   724.4 1903.52   742.3 1906.35
#Mann= 3 ,-1 , 0
       0      .1       0   275.4    .045       0   326.7      .1       0
#XS Ineff= 2 , 0
                           355.3         1742.21
Permanent Ineff=
       F       F
Bank Sta=275.4,326.7
XS Rating Curve= 0 ,0
Exp/Cntr(USF)=0,0
Exp/Cntr=0.3,0.1

Type RM Length L Ch R = 1 ,22529   ,248.1,235.7,218.5
XS GIS Cut Line= 4
1970585.98123643228082.4731332191970746.64491229228002.141295291
1970941.38876181227868.2548987451971172.64708312227695.419732294
#Sta/Elev= 30
       0 1868.27    75.1 1834.67    97.1 1827.33   119.1 1817.39     200 1786.33
   211.8 1779.53   221.2 1771.96   229.4 1762.07   257.3 1736.53   269.2 1730.13
   280.2 1727.85  286.33 1722.74   289.1 1720.83   306.1 1720.38     321 1720.47
  332.721722.742   360.4 1724.41   372.2 1728.12   439.6  1727.3   461.5 1733.59
     478 1743.15   523.1 1773.99   545.9 1793.75     564 1807.61   572.2 1817.32
   580.4 1823.69   604.5 1837.87     628 1848.94   660.8 1866.98   704.7 1887.73
#Mann= 3 ,-1 , 0
       0      .1       0  286.33    .045       0  332.72      .1       0
Bank Sta=286.33,332.72
XS Rating Curve= 0 ,0
Exp/Cntr(USF)=0,0
Exp/Cntr=0.3,0.1
